--- Lt_Crooked_Cr.prj (project) ---

Proj Title=Lt_Crooked_Cr
Current Plan=p02
Default Exp/Contr=0.3,0.1
English Units
Geom File=g02
Flow File=f01
Plan File=p02
Y Axis Title=Elevation
X Axis Title(PF)=Main Channel Distance
X Axis Title(XS)=Station
BEGIN DESCRIPTION:
END DESCRIPTION:
DSS Export Rating Curves= 0
DSS Export Rating Curve Sorted= 0
DSS Export Volume Flow Curves= 0
DXF OffsetX= 0
DXF OffsetY= 0
DXF ScaleX= 1
DXF ScaleY= 10

--- Lt_Crooked_Cr.p02 (plan) ---

Plan Title=Lt_Crooked_Cr
Program Version=3.12
Short Identifier=LDS
Geom File=g02
Flow File=f01
Subcritical Flow
K Sum by GR= 0
Std Step Tol= 0.01
Critical Tol= 0.01
Num of Std Step Trials= 20
Max Error Tol= 0.3
Flow Tol Ratio= 0.001
Split Flow NTrial= 30
Split Flow Tol= 0.02
Split Flow Ratio= 0.02
Log Output Level= 0
Friction Slope Method= 1
Unsteady Friction Slope Method= 2
Unsteady Bridges Friction Slope Method= 1
Parabolic Critical Depth
Global Vel Dist= 0 , 0 , 0
Global Log Level= 0
CheckData=True
Encroach Param=-1 ,0,0, 2
Encroach River=Lt_Crooked_Cr
Encroach Reach=Main
Encroach Node=15213.53
       1459.4183     580
Encroach Node=15015.91
       1     322     360
Encroach Node=14888.24
       1     310     419
Encroach Node=14854.35
       1     310420.8014
Encroach Node=14567.31
       1  363.64429.2188
Encroach Node=14070.2
       1  489.32580.9405
Encroach Node=13870.76
       1  362.78421.8836
Encroach Node=13628.78
       1     195344.7971
Encroach Node=13591.64
       1     170     300
Encroach Node=13338.32
       1  450.81523.1506
Encroach Node=13046.58
       1     344  378.42
Encroach Node=12837.97
       1     202     265
Encroach Node=12532.81
       1     600746.3853
Encroach Node=12359.14
       1     340     403
Encroach Node=12226.4
       1     392   440.8
Encroach Node=12137.75
       1     389   429.7
Encroach Node=11712.69
       1374.7446  447.05
Encroach Node=10884.68
       1 608.988     714
Encroach Node=10249.15
       1     740     971
Encroach Node=9466.78
       1     480     650
Encroach Node=9116.096
       1     328     549
Encroach Node=9056.125
       1     348     513
Encroach Node=8543.376
       1     580 824.402
Encroach Node=7935.252
       1938.44511055.813
Encroach Node=7259.751
       1649.3222  868.22
Encroach Node=6816.38
       1     820     950
Encroach Node=6252.28
       1     700     800
Encroach Node=5938.844
       1     410823.6094
Encroach Node=5875.813
       1     410     800
Encroach Node=5616.38
       1274.3683     500
Encroach Node=5327.802
       1284.1611     400
Encroach Node=5025.465
       1264.2784596.2574
Encroach Node=4956.814
       1     323     577
Encroach Node=4747.213
       1  410.05  463.88
Encroach Node=4345.773
       1 540.524  626.79
Encroach Node=3844.177
       1  669.01743.1189
Encroach Node=3120.083
       1789.14121044.326
Encroach Node=2301.944
       1  707.74883.1046
Encroach Node=1636.742
       11737.2522036.169
Encroach Node=857.834
       1   560.7     680
Encroach Node=697.773
       1     585     729
Encroach Node=429.53
       1     450834.6926
Encroach Node=174.158
       1    12632079.294
Computation Interval=1HOUR
Output Interval=1HOUR
Run HTab= 0
Run UNet= 0
Run PostProcess= 0
UNET Theta= 1
UNET Theta Warmup= 1
UNET ZTol= 0.02
UNET ZSATol= 0.05
UNET MxIter= 20
UNET MaxInSteps= 0
UNET DtIC= 0
UNET DtMin= 0
UNET MaxCRTS= 20
UNET WFStab= 2
UNET SFStab= 1
UNET WFX= 1
UNET SFX= 1
UNET DSS MLevel= 4
UNET DZMax Abort= 100
UNET Convert EG Bridges=-1
UNET Use Existing IB Tables=-1
UNET Froude Reduction=False
UNET Froude Limit= 1
UNET Froude Power= 10
Instantaneous Interval=1HOUR
Write IC File= 0
Echo Input=False
Echo Output=False
Write Detailed= 0
Detailed Automatic Start=False, 10

--- Lt_Crooked_Cr.f01 (steady flow) ---

Flow Title=Lt_Crooked_Cr
Program Version=3.12
Number of Profiles= 2
Profile Names=P100yr,enc
River Rch & RM=Lt_Crooked_Cr,Main            ,15213.53
    1330    1330
River Rch & RM=Lt_Crooked_Cr,Main            ,13870.76
    1530    1530
River Rch & RM=Lt_Crooked_Cr,Main            ,13628.78
    1680    1680
River Rch & RM=Lt_Crooked_Cr,Main            ,9466.78
    1835    1835
River Rch & RM=Lt_Crooked_Cr,Main            ,7259.751
    2280    2280
River Rch & RM=Lt_Crooked_Cr,Main            ,3120.083
    2650    2650
River Rch & RM=Lt_Crooked_Cr,Main            ,857.834
    2960    2960
Boundary for River Rch & Prof#=Lt_Crooked_Cr,Main            , 1
Up Type= 0
Dn Type= 3
Dn Slope=0.0008
DSS Import GetInterval= 0
DSS Import GetPeak= 0
DSS Import FillOption= 0

--- Lt_Crooked_Cr.g02 (geometry) ---

Geom Title=Lt_Crooked_Cr
Program Version=3.12

River Reach=Lt_Crooked_Cr   ,Main
Reach XY= 30
   1046890.22318   680387.739235   1047250.30584   680663.498474
  1047535.129398   680580.005642  1047842.751291   680686.309121
  1047869.309743   680606.559977   1048051.63091   680583.749369
  1048373.441358   680957.878017  1048882.381627   681322.438407
  1049246.999379    680895.18874  1049725.498163   681012.940534
  1049881.129807   680971.132679  1050393.879359   680186.941187
  1050644.501316   680035.000065   1051069.87912   680069.189354
  1051274.998584    680164.13054  1051690.251065   681134.628604
  1051905.381168   681088.880394  1051985.130312   681366.130437
  1052562.379604    682036.43674  1053200.380754    682537.68881
   1054681.49844   683466.252025  1055087.878996    684020.75211
  1056425.628485   684697.190136  1056862.380854   684659.248886
  1057238.000459   684380.692202  1057230.377816   684181.999344
  1057467.249485   684008.812284  1057610.130249   683431.558914
  1057576.629058   683346.501374  1057449.128769   683344.940782

Type RM Length L Ch R = 1 ,15213.53,208.01,197.61,186.28
XS GIS Cut Line= 3
  1047001.189988   681107.105268  1047221.115696   680579.732391
  1047324.346109   680193.740348
#Sta/Elev= 30
       0 1580.58   74.72 1566.66   97.14 1564.16  114.94 1563.22  132.81 1564.16
  196.31 1560.85  215.39 1558.09  361.56 1551.16  379.99 1543.04  394.81 1541.28
  433.99 1539.84  451.79 1536.88  484.41 1535.26  488.26 1531.66  489.93 1530.24
  495.02 1529.24  505.84 1531.34  522.23 1534.01  554.92 1535.63  603.73 1536.07
  685.51 1539.89  721.54 1542.52  743.13 1546.22  764.75 1552.36  805.68  1566.3
   839.6  1582.3  878.92 1596.32  894.52 1603.12  917.87 1614.22  970.95  1645.6
#Mann= 3 , 0 , 0
       0      .1       0  488.26    .045       0  505.84      .1       0
Bank Sta=488.26,505.84
Exp/Cntr=0.3,0.1

Type RM Length L Ch R = 1 ,15015.91,124.87,127.68,130.18
XS GIS Cut Line= 3
  1047373.226997   680968.140547  1047383.046058   680626.928296
  1047385.500814   680236.620741
#Sta/Elev= 30
       0 1580.39    8.52  1577.8   40.78 1572.54   76.63  1564.4  138.45  1552.8
  152.25 1548.98  168.78 1542.64  172.66 1540.69  193.68  1540.1  219.09 1536.63
  253.12 1533.85  315.75 1531.73  326.87 1530.17  339.54  1528.1  345.64 1529.06
  351.74 1530.97  367.19 1532.43  383.78 1533.12  400.28 1532.71  455.73 1536.36
  467.51 1537.73  479.54 1539.52  492.36 1542.71  513.19 1550.39  535.69 1554.84
   558.3 1557.23  567.47 1559.38  582.82 1568.46  635.34 1589.88  731.67  1632.4
#Mann= 3 , 0 , 0
       0      .1       0  326.87    .045       0  351.74      .1       0
#Block Obstruct= 1 ,-1
   205.6  240.68 1545.98
Bank Sta=326.87,351.74
Exp/Cntr=0.5,0.3

Type RM Length L Ch R = 1 ,14888.24,34.12,33.89,32.71
BEGIN DESCRIPTION:
Upstream xs of Bridge 37111-0336
END DESCRIPTION:
XS GIS Cut Line= 4
   1047471.84888   680974.701022  1047497.991396   680625.363238
  1047506.547466   680558.747976   1047487.55787   680308.191496
#Sta/Elev= 30
       0  1575.9    42.8  1566.4    76.6  1559.9      83  1557.5   132.3    1550
   147.9  1540.3   171.9    1540   211.7  1534.4   224.7  1533.5   266.9  1532.1
   357.1  1531.7   379.6  1530.3   381.2  1528.5   387.2  1527.1   398.2  1527.8
   399.2  1528.3   400.5  1531.2   437.9  1537.7   455.8  1539.2   470.4  1542.2
   480.9  1543.3     497  1547.7   498.6  1552.1   527.4  1563.7   533.5  1565.5
   546.6  1571.8   560.4  1579.8   589.6  1589.3   638.3  1610.6   668.8  1625.9
#Mann= 3 , 0 , 0
       0      .1       0   379.6    .045       0   400.5      .1       0
#XS Ineff= 2 , 0
       0                   411.2       0  1534.4
Permanent Ineff=
       F       F
Bank Sta=379.6,400.5
Exp/Cntr=0.5,0.3

Type RM Length L Ch R = 3 ,14871.26,,,
BEGIN DESCRIPTION:
Bridge : 37111-0336 (Gravel Rd)
END DESCRIPTION:
Bridge Culvert--1,0,-1,-1, 0
Deck Dist Width WeirC Skew NumUp NumDn MinLoCord MaxHiCord MaxSubmerge Is_Ogee
11,12,2.6,0, 55, 47, , , 0.95, 0, 0,0,,
      -3     2.1     3.4    20.2      21    33.1    44.6      69    84.6    85.5
      92   110.5   122.9   127.2   140.6   155.2   159.4   168.7   175.4   185.9
   191.1   201.6   207.3   216.1   226.4   240.1   241.3   261.6   265.7   276.5
   278.2   281.6   290.4   294.9   304.2   310.2   318.3     331     332   332.9
   333.9   347.3   351.6   380.2   380.2   400.2   400.2   413.6   414.4   415.1
   429.1   440.6   444.3   449.7     456
  1575.9  1574.8  1574.5  1571.4  1571.3    1568  1566.3  1561.6  1558.3  1557.9
  1556.7  1553.5  1551.8  1548.7  1539.7    1540  1540.2  1539.3  1538.8    1537
  1536.1  1534.5  1533.7  1533.3    1533  1532.7  1532.7  1532.3  1532.4  1532.2
  1532.2  1532.2    1532  1532.1    1532  1532.1  1532.2  1532.6  1532.7  1532.6
  1532.7  1533.3  1533.6  1534.5  1534.5  1534.5  1534.5    1535  1535.1  1535.2
  1537.1  1538.5  1538.8  1539.2  1539.6
                                                                                
                                                                                
                                                                                
                                                                                
                                  1532.5  1532.5
                                        
   245.8   246.9   267.3   271.4   282.2   283.9   287.3   296.1   300.6   309.9
   315.9     324   336.7   337.7   338.6   339.6     353   357.3   385.9   385.9
   405.9   405.9   419.3   420.1   420.8   434.8   446.3     450   455.3   461.7
   463.4   486.7   489.2   489.9   492.6     550   562.2     569   571.4   576.1
   591.2   615.7   628.8   632.7     638   654.2   671.4
  1532.3  1532.7  1532.3  1532.4  1532.2  1532.2  1532.2    1532  1532.1    1532
  1532.1  1532.2  1532.6  1532.7  1532.6  1532.7  1533.3  1533.6  1534.5  1534.5
  1534.5  1534.5    1535  1535.1  1535.2  1537.1  1538.5  1538.8  1539.2  1539.6
  1539.7  1544.4  1545.1  1546.3  1553.8  1576.9  1580.5  1583.8  1585.1  1587.9
  1592.8  1603.6  1609.9  1611.2  1615.5    1623  1631.7
                                                                                
                                                                          1532.5
  1532.5
                                                                                
                                                        
BR Coef=-1 , 1 , 0 ,, 0 ,,,0.8,0,1.2,0,
WSPro=,,,, 1 ,,,, 0 ,,,, 0 ,,,,-1 ,-1 ,-1 , 0 , 0 , 0 , 0 , 0
BC Design=,, 0 ,, 0 ,,,,,,

Type RM Length L Ch R = 1 ,14854.35,286.76,287.04,288.64
BEGIN DESCRIPTION:
Down stream xs of Bridge 37111-0336
END DESCRIPTION:
XS GIS Cut Line= 4
  1047504.487791   680974.701022  1047530.630308   680625.363238
  1047539.186378   680558.747976  1047520.196781   680308.191496
#Sta/Elev= 30
       0  1575.2    28.4  1569.8    52.3  1566.2   119.6  1554.2   138.8  1539.9
   157.9  1539.9     191  1536.4   208.4  1533.3   223.6  1532.6   258.4  1531.5
   300.5  1531.2   324.9  1532.3   337.4  1532.1   350.3    1533  382.831529.792
   392.9  1527.1   400.9  1527.2   403.9  1527.8  406.771529.383   430.3  1535.6
     465  1540.8   475.4    1546   481.7  1552.2   495.4  1561.2   567.3  1590.1
   589.2  1597.1     626  1614.9   636.9  1618.6   651.5  1630.4   668.8  1638.5
#Mann= 3 , 0 , 0
       0      .1       0  382.83    .048       0  406.77     .12       0
#XS Ineff= 2 , 0
       0  375.15 1532.12   416.8       0  1532.7
Permanent Ineff=
       F       F
Bank Sta=382.83,406.77
Exp/Cntr=0.5,0.3

Type RM Length L Ch R = 1 ,14567.31,475.07,497.11,507.87
XS GIS Cut Line= 3
  1047736.344897   681068.557941  1047787.343133   680664.214574
  1047827.413225   680391.009589
#Sta/Elev= 30
       0 1581.41   78.75 1575.61  125.91 1569.98   186.9 1558.14  202.81 1553.68
  226.91 1548.19  245.91 1536.52  247.28 1536.27  275.56 1535.59  304.88 1531.13
  336.64 1529.78  352.14  1528.1  373.64 1527.68  385.28 1525.03  391.73 1526.13
  398.09 1528.01  417.62 1528.24  429.61 1531.42  445.97 1540.09   456.3 1549.11
  474.13 1557.85  494.86 1577.84  535.89 1597.97  574.09 1607.03  584.35 1608.77
  621.21 1626.12  629.84 1631.02  654.14 1646.64  670.55 1653.12  683.67 1651.61
#Mann= 3 , 0 , 0
       0      .1       0  373.64    .048       0  398.09     .12       0
Bank Sta=373.64,398.09
Exp/Cntr=0.3,0.1

Type RM Length L Ch R = 1 ,14070.2 ,207.05,199.44,196.15
XS GIS Cut Line= 3
  1047812.842289   681079.486124  1048158.901914   680700.641913
  1048308.253985   680467.506982
#Sta/Elev= 30
       0 1578.22   40.73 1575.95   69.94 1572.57   99.04 1568.12  125.07  1565.4
  158.48 1559.05  214.73 1552.99  229.26 1550.81  280.51 1548.07  302.74 1545.01
  340.45 1536.11  359.54 1529.37  374.44 1531.36  398.94  1531.8  405.69 1531.04
  417.99 1527.51  478.63 1526.73  499.32 1523.97     509 1521.72   521.6 1523.73
  530.64 1525.45  556.03 1525.35   580.3 1528.06  651.58 1551.13  666.15 1549.93
  678.97 1555.28  700.37  1560.8  748.83 1567.34  774.96 1572.16  789.98 1576.41
#Mann= 3 , 0 , 0
       0      .1       0  499.32    .048       0   521.6     .12       0
Bank Sta=499.32,521.6
Exp/Cntr=0.3,0.1

Type RM Length L Ch R = 1 ,13870.76,238.37,241.98,244.89
XS GIS Cut Line= 2
  1048114.019906   681176.836433  1048491.185229   680487.534319
#Sta/Elev= 30
       0 1533.29  202.01 1530.07  227.79 1531.19  257.74 1530.77  283.74 1527.42
   332.6 1525.48  348.56 1525.57  364.35 1524.49  372.78 1522.92  379.01 1521.07
     386 1520.07  399.94 1522.07  411.31 1525.71  427.71  1523.4  442.87 1527.86
  456.65 1526.98   473.5 1533.97  497.03 1542.34  518.08 1545.65  538.95 1550.25
  579.45 1561.83  593.23 1564.39  663.61 1570.74  692.61 1571.99  706.93 1574.54
  726.56 1576.27  738.05 1576.48  748.94 1579.52   763.3 1580.87  785.74 1580.87
#Mann= 3 , 0 , 0
       0      .1       0  372.78    .045       0  399.94     .12       0
Bank Sta=372.78,399.94
Exp/Cntr=0.5,0.3

Type RM Length L Ch R = 1 ,13628.78,37.13,37.14,37.34
BEGIN DESCRIPTION:
Upstream xs of Bridge 37111-0335
END DESCRIPTION:
XS GIS Cut Line= 3
  1048329.599499   681197.754166  1048469.383507   680994.044532
  1048681.501906   680585.985439
#Sta/Elev= 30
       0    1557    51.7  1555.4    68.8  1553.1   100.5    1544   119.7  1529.3
   137.9  1529.1   172.7  1524.1   190.5  1523.7  204.641521.968   210.7  1516.9
   215.7  1516.7   230.7  1517.1   239.7  1521.7   256.4  1524.6   337.3  1525.9
   405.9  1529.1   449.1  1533.1   462.9  1535.6   479.4  1542.4   489.6  1544.7
   509.2    1545   518.7  1543.1   533.4  1542.1     552  1544.4   565.9  1547.3
   602.5  1551.3   615.4  1554.3   631.3  1555.5   683.6  1563.1     707  1563.2
#Mann= 3 , 0 , 0
       0      .1       0  204.64    .045       0   239.7     .12       0
#XS Ineff= 2 , 0
       0     193  1526.4  242.63       0 1525.09
Permanent Ineff=
       F       F
Bank Sta=204.64,239.7
Exp/Cntr=0.5,0.3

Type RM Length L Ch R = 3 ,13615.07,,,
BEGIN DESCRIPTION:
Bridge : 37111-0335 (gravel road)
END DESCRIPTION:
Bridge Culvert--1,0,-1,-1, 0
Deck Dist Width WeirC Skew NumUp NumDn MinLoCord MaxHiCord MaxSubmerge Is_Ogee
7.7,12,2.6,0, 19, 19, , , 0.95, 0, 0,0,,
       0   140.3   147.5   154.6   164.5   168.5   181.6   182.6   187.8   200.7
   200.7   234.7   234.7   242.1   252.4   254.1   259.1     269     500
    1528  1529.1    1529  1527.9  1527.9  1527.5    1527    1527  1526.8  1526.5
  1529.3  1529.3  1526.5  1526.3  1525.4  1525.2  1525.1  1525.4  1524.6
                                                                                
    1524    1524
   153.7   157.7   170.8   171.8     177   189.9   189.9   223.9   223.9   231.3
   241.6   243.3   248.3   258.2   264.1     273   279.8     288   295.6
  1527.9  1527.5    1527    1527  1526.8  1526.5  1529.3  1529.3  1526.5  1526.3
  1525.4  1525.2  1525.1  1525.4    1525  1526.1  1525.8  1525.6  1525.4
                                                    1524    1524
                                                                        
BR Coef=-1 , 1 , 0 ,, 0 ,,,0.8,0,1.2,0,
WSPro=,,,, 1 ,,,, 0 ,,,, 0 ,,,,-1 ,-1 ,-1 , 0 , 0 , 0 , 0 , 0
BC Design=,, 0 ,, 0 ,,,,,,

Type RM Length L Ch R = 1 ,13591.64,259.21,253.32,246.71
BEGIN DESCRIPTION:
Down stream xs of Bridge 37111-0335
END DESCRIPTION:
XS GIS Cut Line= 3
  1048364.545511   681212.243934  1048504.329519     681008.5343
  1048716.447918   680600.475207
#Sta/Elev= 30
       0  1562.6    44.2  1556.8    89.3  1544.1   110.2  1531.8   121.7  1528.9
   148.2  1528.8   165.8  1526.9   173.8  1524.4     194  1521.5   197.5    1520
   197.9  1518.7   199.9  1516.9   204.9  1516.7   219.9  1517.1   221.9  1518.2
   223.2  1520.3   239.6    1526   260.2  1526.7   302.4  1525.6   331.2  1527.6
   359.6  1530.8   389.1  1531.6   433.6  1536.6   462.1  1542.9   490.2  1543.9
   534.1  1555.5   609.3  1562.1   634.8  1566.7   677.1    1572     707  1572.1
#Mann= 3 , 0 , 0
       0    .095       0   197.5    .045       0   223.2     .12       0
#XS Ineff= 2 , 0
       0  172.47 1524.87               0
Permanent Ineff=
       F       F
Bank Sta=197.5,223.2
Exp/Cntr=0.5,0.3

Type RM Length L Ch R = 1 ,13338.32,300.95,291.74,284.99
XS GIS Cut Line= 3
  1048515.667267   681604.184666  1048714.639396    681120.34292
    1048820.3107   680795.200408
#Sta/Elev= 30
       0 1557.71   34.56 1554.23   65.78 1553.76   82.66 1550.98  130.06  1546.6
  154.95 1547.08  199.62 1549.96  215.76 1549.16  233.06 1546.77  258.43 1547.37
  284.71 1545.97  295.53 1544.36  342.38 1530.28  360.64 1528.63  376.02 1528.84
  407.99 1522.73   447.9  1520.9  460.81 1519.32  476.61  1516.9  486.29 1520.46
  498.12 1521.34  527.45 1525.74  541.13 1531.67  554.55 1540.26   601.9 1552.85
  690.13 1566.71  713.88 1568.52  808.25 1584.65  834.45 1587.76  865.04 1592.82
#Mann= 3 , 0 , 0
       0    .095       0  460.81    .045       0  486.29     .12       0
Bank Sta=460.81,486.29
Exp/Cntr=0.3,0.1

Type RM Length L Ch R = 1 ,13046.58,227.6,208.62,183.71
XS GIS Cut Line= 2
  1048901.081817   681668.637531  1048925.362917   680775.632929
#Sta/Elev= 30
       0 1620.49   58.71 1612.86  101.57 1599.82  122.35 1590.79  158.22 1579.92
  180.88  1568.8  189.64 1569.07  217.11 1561.82  257.45 1554.81   263.3 1550.11
   285.8 1538.11  321.48 1535.86  338.85 1527.52  345.59 1518.11  352.65 1515.62
  368.42 1517.78  386.71  1518.4  395.61 1521.28  413.95 1531.34  435.37 1534.62
  447.99 1539.24  473.35 1542.85   514.9 1544.62  524.19 1548.32  563.06 1557.03
  615.56  1559.1  681.91 1565.21  721.66 1573.53  792.32  1592.6  893.33 1611.86
#Mann= 3 , 0 , 0
       0    .095       0  345.59    .049       0  368.42     .12       0
Bank Sta=345.59,368.42
Exp/Cntr=0.3,0.1

Type RM Length L Ch R = 1 ,12837.97,297.86,305.15,311.31
XS GIS Cut Line= 4
  1049118.389463   681384.270453  1049084.841631   681208.144274
   1049042.90682   681147.338822  1049017.745965    680776.21586
#Sta/Elev= 30
       0 1556.77    1.44 1557.23   10.73 1555.92   21.54 1559.36    34.8 1560.17
  139.37 1527.85  157.74 1526.17  168.17 1526.22  177.88  1524.6  209.54 1509.61
  216.28 1507.11  223.03 1506.12     236 1508.14  255.56 1512.37  268.78 1513.99
  270.56 1514.81  283.95  1516.1  297.32  1519.4  334.74 1522.53  353.34 1527.79
  361.94 1532.22  365.89 1533.36  395.92 1540.16  400.66 1541.77  413.01 1542.85
  422.79 1545.23  463.82 1557.56   536.8  1586.7  608.21 1607.85  625.13 1611.62
#Mann= 3 , 0 , 0
       0    .095       0  209.54    .049       0     236     .12       0
Bank Sta=209.54,236
Exp/Cntr=0.3,0.1

Type RM Length L Ch R = 1 ,12532.81,155.85,173.68,191.15
XS GIS Cut Line= 3
  1049235.621318    681649.75221  1049224.829723   680953.694276
  1049141.194828   680743.258143
#Sta/Elev= 30
       0 1614.78   28.63  1610.6   67.47 1601.61  126.78 1590.84  141.78 1585.42
  152.99 1583.42  203.23 1577.19  257.95 1577.31  286.49 1574.33  390.03  1556.1
   433.4 1546.66  446.91 1542.72   462.9  1537.4  478.31 1527.96   526.7 1516.03
  547.68 1512.58  577.63 1509.88  619.64 1509.16   668.9 1505.92   699.2 1506.14
  727.73 1507.92  741.25 1504.81  744.57 1506.36  745.85 1508.24  750.97 1514.91
  772.31 1522.74  824.52 1546.96  841.04 1550.02     886 1567.44  922.59 1579.55
#Mann= 3 , 0 , 0
       0      .1       0  727.73    .049       0  745.85     .12       0
Bank Sta=727.73,745.85
Exp/Cntr=0.3,0.1

Type RM Length L Ch R = 1 ,12359.14,122.7,132.74,142.78
XS GIS Cut Line= 2
  1049294.515643   681302.078244  1049411.933057   680738.055186
#Sta/Elev= 30
       0 1563.17    12.4 1559.94   32.03 1556.91    69.1 1545.92   84.89 1539.43
  103.13 1530.19  143.14 1529.77  152.15 1528.73  163.61 1526.02  169.65 1523.46
  177.79 1518.25  190.98 1515.82  216.34 1515.23   230.2 1512.18  260.27 1510.13
  321.26 1507.37  343.12 1507.31  378.86 1506.01  391.92 1503.97  398.57 1504.95
  400.48 1506.64  405.24 1510.97  419.09 1512.55  438.49 1520.61  481.48 1535.03
   504.7 1545.24   523.9 1551.24  550.44 1561.33  566.11 1564.23  576.12 1564.43
#Mann= 3 , 0 , 0
       0      .1       0  378.86    .049       0  400.48     .12       0
Bank Sta=378.86,400.48
Exp/Cntr=0.5,0.3

Type RM Length L Ch R = 1 ,12226.4 ,88.66,88.64,88.63
BEGIN DESCRIPTION:
Upstream xs of Bridge 37111-0256
END DESCRIPTION:
XS GIS Cut Line= 5
  1049351.490685   681344.123388  1049446.057413   681050.818597
   1049524.29649   680918.621542  1049553.973407   680878.153068
  1049542.760245   680640.147811
#Sta/Elev= 30
       0  1567.7      78  1550.6   105.8  1542.1   124.3  1532.8   139.9  1527.9
   183.6  1527.9   220.6  1522.7   260.4  1513.3   298.7    1512   343.5  1504.9
   372.1  1506.4   377.7  1503.7     395  1502.8   400.3  1499.3   408.3  1497.7
   424.3  1497.7  429.82 1498.52  432.58 1500.46   439.5  1505.9   446.7  1508.7
   468.4  1510.5   480.4  1509.7   503.2  1514.1     512    1514   523.5  1518.6
   566.6    1531   620.8  1543.4     668  1546.3   704.6  1551.5   750.2  1563.1
#Mann= 3 , 0 , 0
       0      .1       0     395    .047       0  432.58     .12       0
#XS Ineff= 2 , 0
       0   391.8 1509.15   440.8       0  1508.9
Permanent Ineff=
       F       F
Bank Sta=395,432.58
Exp/Cntr=0.5,0.3

Type RM Length L Ch R = 2 ,12186.88,,,
BEGIN DESCRIPTION:
Culvert : 37111-0256 (SR-1104)
END DESCRIPTION:
Bridge Culvert--1,0,-1,-1, 0
Deck Dist Width WeirC Skew NumUp NumDn MinLoCord MaxHiCord MaxSubmerge Is_Ogee
9.5,60,2.6,0, 78, 42, , , 0.95, 0, 0,0,,
    -5.3    77.3   127.6   133.6   145.7   205.7   228.3   240.4   244.9   257.6
   262.1   264.3   272.7   275.1   285.8   291.8   292.6   293.6   302.9   305.5
   307.8   308.9   315.9   322.5   323.9   346.8   357.8     393   400.3   400.3
   431.3   431.3   456.1   456.5     462   464.1   476.9   484.2   491.7   496.2
   506.7   515.6     523     526   531.3   535.6   540.9   547.3   556.2   564.7
   567.1   571.4   578.4   583.6   590.8   608.2   609.8   610.4   619.9   622.7
   634.3     639   640.3   647.2     650   656.9   661.2   663.5   672.1   680.6
   683.3   687.9   704.6   711.3   712.8   725.6   726.1   740.4
    1566  1545.2    1530  1527.7  1526.7  1519.4    1516  1513.8  1513.1  1512.1
    1512  1511.8  1511.6  1511.6  1511.1  1510.9  1510.9  1510.8  1510.5  1510.5
  1510.5  1510.5  1510.4  1510.4  1510.3  1509.5  1509.5  1509.1  1509.5  1509.5
  1509.5  1509.5    1509    1509  1508.9  1508.9  1508.9  1508.8  1508.8  1508.9
  1509.4  1510.2  1510.8  1511.1  1511.2  1511.3  1511.7  1513.1    1515  1517.7
  1518.3    1519  1522.5  1524.6  1528.4  1531.3  1531.8    1532  1535.8  1536.2
  1537.3  1537.5  1537.5  1538.6  1539.2  1539.2  1539.1  1539.1  1539.8  1540.2
  1540.1  1540.9  1543.2  1544.4  1544.7    1547  1547.1  1549.5
                                                                                
                                                                                
                                                                                
                                                                                
                                                                                
                                                                                
                                                                                
                                                                
   300.3   307.3   313.9   315.4   322.7   328.5   332.3   338.2   343.2   349.2
   353.7   357.7     366   369.2   372.2   382.4   384.4   391.8   391.8   422.8
   422.8   447.6   447.9   453.5   455.5   468.3   475.7   483.2   487.6   498.1
     507   514.4   517.4   522.7     527   532.3   538.7   547.6   556.2   558.6
   562.8     660
  1510.5  1510.4  1510.4  1510.3    1510  1509.9  1509.8  1509.5  1509.6  1509.5
  1509.2  1509.4  1509.3  1509.2  1509.3  1509.2  1509.1  1509.5  1509.5  1509.5
  1509.5    1509    1509  1508.9  1508.9  1508.9  1508.8  1508.8  1508.9  1509.4
  1510.2  1510.8  1511.1  1511.2  1511.3  1511.7  1513.1    1515  1517.7  1518.3
    1519 1525.05
                                                                                
                                                                                
                                                                                
                                                                                
                
BR Coef=-1 , 0 , 0 ,, 0 ,,,0.8,-1,,0,
WSPro=,,,, 1 ,,,, 0 ,,,, 0 ,,,,-1 ,-1 ,-1 , 0 , 0 , 0 , 0 , 0
Multiple Barrel Culv=4,8.5,14,60,0.024,0.5,1,29,1,1497.7,1497.7, 2,Culvert #1  , 0 ,9.5
   408.3   399.8   424.3   415.8
Culvert Bottom n=0.024
BC Design=,, 0 ,, 0 ,,,,,,

Type RM Length L Ch R = 1 ,12137.75,464.2,425.06,385.73
BEGIN DESCRIPTION:
Down stream xs of Bridge 37111-0256
END DESCRIPTION:
XS GIS Cut Line= 5
  1049440.521358   681363.008709  1049535.088086   681069.703918
  1049613.327164   680937.506863  1049643.004081   680897.038389
  1049618.638667   680665.440593
#Sta/Elev= 30
       0  1551.6    11.1  1550.3    74.8  1538.4    90.9  1532.4   143.2  1521.2
   164.2    1519   213.3  1517.8   261.4  1514.4   296.2  1515.4   309.9  1513.5
   321.8    1510   367.1  1509.4   386.9  1505.3  391.02 1500.28   391.8  1499.3
   399.8  1497.7   415.8  1497.7   422.8  1499.3   431.2  1504.1   435.9    1504
   442.2  1505.8   464.6    1504     508  1504.1   572.8  1507.5   601.1  1514.9
   638.1  1516.7   656.8  1525.6   676.4  1531.3   711.1  1533.7   744.9  1538.5
#Mann= 3 , 0 , 0
       0    .095       0  391.02     .05       0   422.8    .085       0
#XS Ineff= 2 , 0
       0                   441.9       0  1506.4
Permanent Ineff=
       F       F
Bank Sta=391.02,422.8
Exp/Cntr=0.5,0.3

Type RM Length L Ch R = 1 ,11712.69,816.88,828.01,838.23
XS GIS Cut Line= 3
  1050263.605159    681196.58947  1049939.014198   680859.352099
  1049660.793329    680593.77764
#Sta/Elev= 30
       0 1539.16   27.63 1537.45    44.6 1535.17   80.83 1528.32  122.64 1523.21
  135.38 1520.23  158.59 1517.54  184.74 1512.78   212.8 1511.45  226.32 1507.07
  232.07 1507.55  319.46 1501.78  369.55 1500.53  388.71 1497.35  396.23 1497.44
  413.01 1495.15  426.09  1492.9  437.05 1495.85  448.23 1498.39  483.87 1499.34
  541.52 1498.27  622.63 1501.55  660.72 1504.77  674.47 1504.78  751.03 1521.38
  775.02 1522.81  789.04 1526.13  808.67 1534.06  816.79 1536.18  852.69 1542.98
#Mann= 3 , 0 , 0
       0    .085       0  413.01    .049       0  437.05    .085       0
Bank Sta=413.01,437.05
Exp/Cntr=0.3,0.1

Type RM Length L Ch R = 1 ,10884.68,617.99,635.53,650.99
XS GIS Cut Line= 3
  1050680.409493   680825.101409  1050364.249472   680150.626666
  1050148.206758   679866.082612
#Sta/Elev= 30
       0 1513.89   22.57 1514.59   34.52 1513.57   58.44 1509.63  112.75 1505.96
  210.99 1500.95  353.55 1495.69   587.5    1492  645.28 1491.94  664.33 1492.89
  678.39 1491.15  693.83 1489.14  701.14  1490.2  705.96 1491.62  708.72 1492.52
  721.26 1494.06  809.43 1493.67   862.6 1494.79  884.32 1495.99  902.13 1505.08
  932.59 1506.59  939.83 1507.59  953.45 1516.87  962.15 1521.29  987.48 1526.73
  1019.3 1529.22 1042.71 1533.72 1068.67 1536.44  1087.2 1536.66 1102.17 1538.25
#Mann= 3 , 0 , 0
       0    .085       0  678.39    .049       0  705.96    .085       0
#Block Obstruct= 1 ,-1
  714.74  874.06 1503.26
Bank Sta=678.39,705.96
Exp/Cntr=0.3,0.1

Type RM Length L Ch R = 1 ,10249.15,752.06,782.37,801.83
XS GIS Cut Line= 3
  1050854.297546   680840.909432  1050954.414892   680045.239954
  1051033.387041   679418.118169
#Sta/Elev= 30
       0 1518.25   27.87 1513.71   53.58 1513.27   67.19 1509.17   78.42 1507.96
  119.96 1505.72  382.11  1496.6  545.67 1493.03  648.68 1488.41  689.79 1487.43
  730.11 1488.13  742.01  1486.7  755.46 1483.87  767.76 1486.03  785.99  1487.6
  921.73 1487.37  1139.7 1491.59 1171.56 1493.52 1179.17 1497.52  1196.2 1502.24
 1234.58 1504.08 1242.65 1510.38 1263.66 1520.52 1301.27 1524.55  1319.9 1538.33
    1332 1543.23 1341.24    1546 1355.23 1547.29 1384.83 1557.63 1434.02 1578.06
#Mann= 3 , 0 , 0
       0    .085       0  742.01    .049       0  767.76    .085       0
Bank Sta=742.01,767.76
Exp/Cntr=0.3,0.1

Type RM Length L Ch R = 1 ,9466.78 ,346.8,350.68,354.43
XS GIS Cut Line= 3
  1050961.133429   680868.351367  1051435.942857   680481.278436
   1052251.37648   680145.815256
#Sta/Elev= 30
       0 1527.36   27.53 1524.73   76.24 1512.75  112.75 1512.76  184.41  1504.2
  290.95 1499.07  426.02 1486.56  520.03 1483.75  534.21 1482.19  541.17 1478.32
  548.27 1477.96  571.82  1480.8  588.05 1482.62  677.29 1482.14   850.4  1485.2
  967.39 1489.98 1037.92 1495.33 1053.18 1500.35 1096.76 1505.61 1110.67 1505.82
 1125.18 1507.65 1157.24 1518.34 1171.52 1519.33 1204.01 1524.29 1255.84 1533.43
 1292.86 1535.73 1337.47 1542.21 1382.16 1544.83 1467.54 1543.75 1494.33 1546.45
#Mann= 3 , 0 , 0
       0     .12       0  534.21    .049       0  571.82    .085       0
Bank Sta=534.21,571.82
Exp/Cntr=0.5,0.3

Type RM Length L Ch R = 1 ,9116.096,59.69,59.97,60.71
BEGIN DESCRIPTION:
Upstream xs of Bridge 37111-0254
END DESCRIPTION:
XS GIS Cut Line= 2
  1051254.078131   681010.871305  1051887.638057   680611.125128
#Sta/Elev= 30
       0  1526.1    38.9  1519.7    95.8  1507.3   108.8  1501.4   113.1    1498
   125.9  1496.6   139.2  1497.3   145.6  1496.9   191.5  1490.9   225.9  1487.3
   232.7    1486   282.2  1482.8   323.2  1481.1   330.9  1479.8     339    1475
     355  1472.9  358.721475.203   390.6  1480.5   402.8  1480.1     430  1481.3
   505.2  1481.7   554.1  1483.4   574.3  1484.4   578.8  1485.3   617.8  1485.9
   641.6  1487.6   653.6  1487.5   686.2  1493.6   723.5  1510.1   749.1  1516.3
#Mann= 3 , 0 , 0
       0     .12       0     339    .049       0  358.72    .095       0
#XS Ineff= 2 , 0
       0                   382.7       0  1480.4
Permanent Ineff=
       F       F
Bank Sta=339,358.72
Exp/Cntr=0.5,0.3

Type RM Length L Ch R = 3 ,9086.438,,,
BEGIN DESCRIPTION:
Bridge : 37111-0254 (Cherry Springs Rd.)
END DESCRIPTION:
Bridge Culvert--1,0,-1,-1, 0
Deck Dist Width WeirC Skew NumUp NumDn MinLoCord MaxHiCord MaxSubmerge Is_Ogee
23.7,12,2.6,0, 12, 41, , , 0.95, 0, 0,0,,
   314.7   321.2   330.8     338     338     359     359   387.4   394.1   401.4
   450.3   493.1
  1481.6  1481.3  1480.6  1480.5  1480.5  1480.5  1480.5    1481  1481.1  1481.1
  1480.8  1481.4
                                  1478.7  1478.7
                
   309.1   320.8   324.6   331.1   340.6     348     348     369     369   397.3
     404   454.7   536.3   546.4   550.2   560.8   564.5   575.7     579   590.3
   593.3     605   607.9   620.6   631.2   636.3     646   655.3   660.7   665.4
   666.2   681.2   682.7   692.6   698.8   704.3     711   736.2   739.7   741.1
     745
  1482.2    1482  1481.6  1481.3  1480.6  1480.5  1480.5  1480.5  1480.5    1481
  1481.1  1480.8  1482.7  1483.1  1483.2  1483.6    1484    1485  1485.1  1485.4
  1485.5  1485.7  1486.2  1487.7  1488.5  1489.4  1490.7  1491.3  1491.8  1492.7
    1493  1497.4  1498.1    1503  1505.9  1508.9  1511.1  1518.8  1520.6  1521.4
  1522.9
                                                  1478.7  1478.7
                                                                                
                                                                                
                                                                                
        
BR Coef=-1 , 1 , 0 ,, 0 ,,,0.75,-1,1.2,0,
WSPro=,,,, 1 ,,,, 0 ,,,, 0 ,,,,-1 ,-1 ,-1 , 0 , 0 , 0 , 0 , 0
BC Design=,, 0 ,, 0 ,,,,,,

Type RM Length L Ch R = 1 ,9056.125,521.35,512.75,502.37
BEGIN DESCRIPTION:
Down stream xs of Bridge 37111-0254
END DESCRIPTION:
XS GIS Cut Line= 3
  1051279.219374   681061.153829  1051597.837025   680864.630165
  1051909.008154   680691.456697
#Sta/Elev= 30
       0  1521.5    52.7    1512    89.6  1506.4   101.7  1503.7   111.7    1497
   124.2  1492.8   139.2  1494.1   164.5  1493.5   228.4  1486.1   340.9  1480.5
   347.8  1477.9     349    1475     365  1472.9     368  1474.7   368.6  1478.9
   372.7  1477.4     385  1477.6   403.6  1480.1   447.6  1479.6   490.5  1480.4
   560.7  1483.4   578.4  1485.9   600.5  1487.4   650.4  1493.9     677  1503.2
   695.4  1512.6   710.7  1518.9   716.4  1519.3   722.9  1521.7   730.5  1525.8
#Mann= 3 , 0 , 0
       0    .085       0     349    .049       0     368    .095       0
#XS Ineff= 2 , 0
       0                   393.3       0  1478.9
Permanent Ineff=
       F       F
Bank Sta=349,368
Exp/Cntr=0.5,0.3

Type RM Length L Ch R = 1 ,8543.376,597.84,608.12,607.76
XS GIS Cut Line= 3
  1051399.816071   681697.719595  1051890.108424    681073.24197
  1052070.742433   680928.734747
#Sta/Elev= 30
       0 1508.35   43.35 1506.88   87.46 1504.01  142.96 1499.07  248.35 1487.22
  274.55  1486.7  295.94 1484.55  338.38 1482.78  393.37 1482.18  417.03 1480.65
  460.24  1480.4  493.19 1478.72  602.19 1476.88  650.39  1478.1  688.12 1477.93
  774.58  1474.7  788.36 1472.28     795 1473.48  802.01 1476.34  812.09 1476.79
  826.43 1480.12  843.36 1481.52  860.11 1484.86  873.31 1489.33  890.59  1498.1
  899.04 1503.62  942.34 1522.59  983.77 1533.12 1011.67 1538.52 1025.28 1539.41
#Mann= 3 , 0 , 0
       0    .085       0  774.58    .049       0  802.01     .12       0
Bank Sta=774.58,802.01
Exp/Cntr=0.3,0.1

Type RM Length L Ch R = 1 ,7935.252,685.68,675.5,657.2
XS GIS Cut Line= 3
  1051389.494121   682202.462647  1052036.196977   681651.378241
  1052411.082735   681375.610652
#Sta/Elev= 30
       0 1545.95   22.45 1546.16   78.11 1544.47  145.41 1545.19  188.29 1543.34
  281.23 1541.96  342.55 1538.19  436.93 1523.67  521.26 1507.45  556.01 1498.78
  566.13    1492  575.44 1490.12  590.45 1490.85  598.07 1490.47  608.49  1487.6
  650.61 1483.89  702.15 1481.42  760.51 1477.45  888.71 1475.66  927.18 1473.43
  981.27 1474.14 1001.81 1475.04  1014.6 1471.82 1030.67 1474.73 1052.05 1475.53
 1116.33 1514.64 1162.67 1541.68 1201.66 1562.86 1260.28  1598.5 1315.05 1629.96
#Mann= 3 , 0 , 0
       0    .085       0 1001.81    .049       0 1030.67     .12       0
Bank Sta=1001.81,1030.67
Exp/Cntr=0.3,0.1

Type RM Length L Ch R = 1 ,7259.751,435.6,443.37,449.89
XS GIS Cut Line= 3
  1052189.444819   682785.652511  1052581.678686   682047.633513
  1052793.278544   681614.111846
#Sta/Elev= 30
       0 1495.05    6.24 1492.29   34.22 1492.36   60.21 1498.82   90.63 1501.46
  258.64 1499.97  389.81 1502.55  427.51 1499.04     475 1492.11  561.42 1491.85
  598.75 1485.65  630.41 1476.94  642.35 1475.54  763.92  1471.2  809.76 1472.12
  828.29  1468.7  843.65 1466.67  858.22 1469.84  930.59 1485.03  941.91 1489.11
  988.91 1490.07  999.82 1493.05 1051.46 1526.82 1071.51 1532.64 1100.73 1544.44
 1162.15 1574.65 1182.89    1589 1220.43 1610.58 1306.96 1675.67 1318.18 1681.54
#Mann= 3 , 0 , 0
       0     .09       0  828.29    .049       0  858.22     .12       0
Bank Sta=828.29,858.22
Exp/Cntr=0.3,0.1

Type RM Length L Ch R = 1 ,6816.38 ,571.41,564.1,550.56
XS GIS Cut Line= 3
  1052333.435909   682938.417308  1052921.052084   682294.967524
  1053209.059313   681942.526809
#Sta/Elev= 30
       0  1491.7   14.11 1491.78   41.39 1485.66   92.88 1482.47  237.73 1479.82
  388.87 1481.89  484.79 1481.02  549.57  1482.5  638.38 1476.44   695.6 1473.74
  841.53  1469.5  855.95 1467.89  863.46 1465.67  871.39 1464.68  886.86  1467.3
  919.15 1471.71  943.56 1470.25  955.11 1470.41 1009.79 1472.79 1036.19 1472.97
 1084.77 1475.78 1135.52 1480.62  1182.4 1490.58 1198.21 1492.16 1213.53 1492.37
  1223.4 1494.84  1244.3  1508.3 1252.74 1511.93 1301.55 1538.31 1326.54 1554.29
#Mann= 3 , 0 , 0
       0    .085       0  855.95    .049       0  886.86    .085       0
Bank Sta=855.95,886.86
Exp/Cntr=0.3,0.1

Type RM Length L Ch R = 1 ,6252.28 ,314.34,313.44,308.85
XS GIS Cut Line= 3
  1053075.583733   683299.685325  1053369.759152   682546.183403
  1053571.037061      682066.213
#Sta/Elev= 30
       0 1483.23   77.24 1479.43  227.46 1475.23  466.16 1471.05  616.94 1469.93
  692.09 1467.34  718.75 1462.17   726.2 1463.34  731.65 1461.27   738.3  1460.1
   751.6 1462.08  776.08 1463.54   804.6 1467.85  826.82 1468.85  957.75 1469.45
 1049.99 1471.36 1076.42 1474.08 1091.21 1473.67 1105.89 1475.44 1113.41 1475.35
 1155.98 1483.19 1184.02 1485.16 1191.34 1484.66 1206.39 1487.08  1222.8 1496.78
 1235.07 1501.91 1265.13 1513.13 1276.22 1516.27 1308.36 1529.13 1329.36 1536.42
#Mann= 3 , 0 , 0
       0    .085       0   726.2    .049       0   751.6    .085       0
Bank Sta=726.2,751.6
Exp/Cntr=0.5,0.3

Type RM Length L Ch R = 1 ,5938.844,61.58,63.03,64.32
BEGIN DESCRIPTION:
Upstream xs of Bridge 37111-0246
END DESCRIPTION:
XS GIS Cut Line= 3
  1053446.566535   683241.497896  1053611.717657   682725.400668
  1053760.019016   682313.785931
#Sta/Elev= 30
       0  1491.2    27.3  1487.4    54.4  1486.5    67.6  1484.3   122.5  1480.2
   133.8  1478.3   184.2  1475.7   211.9  1473.4   467.4  1466.7   478.8  1467.3
  496.681464.304   501.6  1462.2     503  1462.5     510    1460     518  1460.1
     521  1461.4     524  1461.5  531.151463.486     551  1466.6   573.7  1467.7
   618.5  1467.2     718    1469   802.3  1469.3   900.7  1472.1   917.5  1474.2
     927  1474.6   936.7  1476.5   951.8  1480.8   974.6    1484   979.4  1485.3
#Mann= 3 , 0 , 0
       0    .085       0  496.68    .049       0  531.15    .085       0
#XS Ineff= 2 , 0
       0   475.6  1468.9   548.4       0  1468.9
Permanent Ineff=
       F       F
Bank Sta=496.68,531.15
Exp/Cntr=0.5,0.3

Type RM Length L Ch R = 3 ,5908.399,,,
BEGIN DESCRIPTION:
Bridge : 37111-0246 (Gravel Road)
END DESCRIPTION:
Bridge Culvert--1,0,-1,-1, 0
Deck Dist Width WeirC Skew NumUp NumDn MinLoCord MaxHiCord MaxSubmerge Is_Ogee
24.4,12,2.6,0, 16, 16, , , 0.95, 0, 0,0,,
       0    69.5   168.9   268.7   368.4     460   466.4     500     500     524
     524     665   760.7   860.6   964.5   979.4
  1493.2    1487  1477.4  1472.8  1470.4  1469.2  1468.9    1469    1469    1469
    1469  1468.8  1469.5  1471.2  1482.3  1486.7
                                                                  1467.2  1467.2
                                                
    -6.1    63.4   162.8   262.6   360.8   424.7   460.3   490.8   490.8   514.8
   514.8   658.9   754.6   854.6   958.4   973.3
  1493.2    1487  1477.4  1472.8  1470.4  1469.2  1468.9    1469    1469    1469
    1469  1468.8  1469.5  1471.2  1482.3  1486.7
                                                                  1467.2  1467.2
                                                
BR Coef=-1 , 1 , 0 ,, 0 ,,,0.8,0,1.2,0,
WSPro=,,,, 1 ,,,, 0 ,,,, 0 ,,,,-1 ,-1 ,-1 , 0 , 0 , 0 , 0 , 0
BC Design=,, 0 ,, 0 ,,,,,,

Type RM Length L Ch R = 1 ,5875.813,252.58,259.43,267.04
BEGIN DESCRIPTION:
Down stream xs of Bridge 37111-0246
END DESCRIPTION:
XS GIS Cut Line= 3
   1053505.25996   683259.105897  1053670.411082   682743.008669
  1053818.712441   682331.393931
#Sta/Elev= 30
       0  1495.9    10.7  1494.8    37.3  1489.5    53.2  1488.5    79.3  1488.6
   103.8  1485.1   130.1  1483.6   171.7  1477.7   209.4  1474.2   308.5  1470.4
   437.2  1468.4   473.6    1467  485.041465.683     493  1462.3   500.8    1460
   508.8  1460.1  516.451463.577   522.2  1463.6   538.5  1466.1   547.2  1466.6
   647.3  1467.3   712.4  1468.6   777.7  1468.2   806.5  1469.3     869    1470
   894.5  1471.1   927.1  1473.6   937.1  1475.4   969.2  1486.7   979.4  1489.6
#Mann= 3 , 0 , 0
       0    .085       0  485.04    .049       0  516.45    .085       0
#XS Ineff= 2 , 0
       0   464.2  1467.4   541.4       0  1467.4
Permanent Ineff=
       F       F
Bank Sta=485.04,516.45
Exp/Cntr=0.5,0.3

Type RM Length L Ch R = 1 ,5616.38 ,281.27,288.58,295.15
XS GIS Cut Line= 3
  1053673.952901   683247.670825  1053851.112277   682939.422971
  1054169.912225   682440.636452
#Sta/Elev= 30
       0 1491.95   10.03 1489.34    40.3 1490.07   59.22  1488.4   71.98  1485.3
   82.27  1484.2   85.35 1483.12  102.63 1480.29  110.12 1478.06   143.7 1474.01
  167.02 1472.22  223.09 1469.35  325.39 1467.39  339.47 1465.53  343.83 1462.21
   347.6 1459.63  355.53 1458.54  371.08 1460.42  395.85 1465.67   407.8 1466.26
  447.18 1465.04  486.62 1465.09  573.79  1467.1  661.33  1467.6  739.66 1467.19
  783.48 1468.04  835.08 1470.65  859.34 1472.88  904.31 1483.83  947.49 1502.08
#Mann= 3 , 0 , 0
       0    .085       0  343.83    .049       0  371.08    .085       0
Bank Sta=343.83,371.08
Exp/Cntr=0.3,0.1

Type RM Length L Ch R = 1 ,5327.802,289.59,302.34,312.81
XS GIS Cut Line= 2
  1053867.026323   683336.068818  1054538.902461   682636.002023
#Sta/Elev= 30
       0 1495.25   22.05  1492.5   33.26 1486.84   56.54 1487.36   75.27 1486.05
   89.57 1482.41  199.94 1473.06  271.93 1468.42  286.43  1465.9  291.74 1460.54
  293.38 1458.99  301.35    1458  317.74 1460.01  344.08 1464.49  357.56 1465.05
  404.82 1464.57  468.76  1466.3   500.4 1465.37  676.22 1465.76  791.39  1468.6
  824.41 1470.36  845.03 1472.54  855.07  1474.8     873 1476.28  899.96 1480.95
   916.1 1489.67  922.56 1490.52  933.43 1490.94   942.8 1489.74  970.31 1490.73
#Mann= 3 , 0 , 0
       0    .085       0  291.74    .049       0  317.74    .085       0
Bank Sta=291.74,317.74
Exp/Cntr=0.5,0.3

Type RM Length L Ch R = 1 ,5025.465,69.7,68.65,67.33
BEGIN DESCRIPTION:
Upstream xs of Bridge 37111-0242
END DESCRIPTION:
XS GIS Cut Line= 3
  1053979.867984   683429.301214  1054393.630943   683232.042148
  1054663.057986   683162.279759
#Sta/Elev= 30
       0  1491.9    13.5  1491.1    23.5  1489.3    35.6  1485.7    49.4  1485.7
    74.7  1481.6   102.4  1482.1   127.8  1475.9   149.2  1473.8   239.4  1468.3
   277.9  1464.5   304.8  1462.7   358.8  1460.5  368.711458.999   390.7  1457.3
   398.7  1458.6   402.1    1460     406  1460.6   412.5  1462.1   426.2  1462.8
   432.1  1463.8   491.4    1464   531.8  1463.4   587.1    1465   601.2  1466.3
   615.6  1469.5   659.1  1488.6     684  1503.3   702.4  1517.7   736.7  1535.7
#Mann= 3 , 0 , 0
       0    .085       0  368.71    .049       0     406     .09       0
#XS Ineff= 2 , 0
       0   333.2  1465.3               0
Permanent Ineff=
       F       F
Bank Sta=368.71,406
Exp/Cntr=0.5,0.3

Type RM Length L Ch R = 3 ,4988.955,,,
BEGIN DESCRIPTION:
Bridge : 37111-0242 (Gravel Rd.)
END DESCRIPTION:
Bridge Culvert--1,0,-1,-1, 0
Deck Dist Width WeirC Skew NumUp NumDn MinLoCord MaxHiCord MaxSubmerge Is_Ogee
30.5,12,2.6,0, 38, 38, , , 0.95, 0, 0,0,,
     100     202   207.5   214.9   221.1     228   232.9   237.9   245.4   251.4
     258   264.8   270.6   278.3   283.2   291.8     296   305.6   308.8   319.2
   321.5   333.2   334.7   346.7   355.6   363.7   363.7   410.7   410.7   441.2
   453.9   458.6   467.5   476.9     481   492.7   494.4   497.3
  1474.6  1470.4  1470.3  1469.8  1469.6  1469.1  1469.7  1469.4    1469  1468.7
  1468.3    1468  1467.7  1467.5  1467.3  1467.1  1466.9  1466.8  1466.5  1466.1
    1466  1465.6  1465.6  1465.3  1465.4    1466    1466    1466    1466  1465.3
  1464.7  1464.7  1464.4    1464  1463.9  1463.5  1463.5  1463.5
                                                                                
                                                                                
                                                  1464.6  1464.6
                                                                
   105.3   207.3     212     220   225.5   232.9   239.1     246   250.9   255.9
   263.4   269.4     276   282.8   288.6   296.3   301.3   309.8     314   323.6
   326.8   337.2   339.6   351.2   352.7   364.7   373.6   378.1   381.7   381.7
   428.7   428.7   459.2   471.9   476.6   485.5   494.9     499
  1474.6  1471.8  1471.4  1470.4  1470.3  1469.8  1469.6  1469.1  1469.7  1469.4
    1469  1468.7  1468.3    1468  1467.7  1467.5  1467.3  1467.1  1466.9  1466.8
  1466.5  1466.1    1466  1465.6  1465.6  1465.3  1465.4  1465.4    1466    1466
    1466    1466  1465.3  1464.7  1464.7  1464.4    1464  1463.9
                                                                                
                                                                                
                                                                          1464.6
  1464.6
Pier Skew, UpSta & Num, DnSta & Num=  ,386.9, 2 ,405.6, 2 , 0 , 0 , 0 ,,
       1       1
  1456.5  1465.1
       1       1
  1456.5  1465.1
BR Coef=-1 , 1 , 0 ,, 0 ,,,0.8,0,2,0,
WSPro=,,,, 1 ,,,, 0 ,,,, 0 ,,,,-1 ,-1 ,-1 , 0 , 0 , 0 , 0 , 0
BC Design=,, 0 ,, 0 ,,,,,,

Type RM Length L Ch R = 1 ,4956.814,221.31,209.6,197.58
BEGIN DESCRIPTION:
Down stream xs of Bridge 37111-0242
END DESCRIPTION:
XS GIS Cut Line= 3
  1054017.271198   683479.602108  1054431.034157   683282.343042
    1054700.4612   683212.580653
#Sta/Elev= 30
       0    1493    26.3  1489.2    37.7  1485.6    86.7  1479.8   125.2  1479.5
   132.4  1477.9   144.5  1473.7   148.7  1473.2   199.8  1470.2   344.2  1464.7
   371.7  1463.3  386.411461.396   395.3  1457.5   395.7    1458   408.7  1457.3
  421.871458.998   445.5  1461.5   459.4  1463.7   470.9  1463.5   491.1  1464.7
   522.8  1463.3   554.9  1463.6   592.6  1466.5   640.4  1485.6   652.9  1492.9
   684.9  1517.5   687.6  1520.2   696.3  1526.1   728.1  1542.6   736.7  1545.5
#Mann= 3 , 0 , 0
       0    .085       0  386.41    .049       0  421.87     .09       0
#XS Ineff= 2 , 0
       0   355.5    1465  455.05       0    1464
Permanent Ineff=
       F       F
Bank Sta=386.41,421.87
Exp/Cntr=0.5,0.3

Type RM Length L Ch R = 1 ,4747.213,393.62,401.44,405.07
XS GIS Cut Line= 3
  1054264.922151   683716.190971  1054591.404238    683360.36219
  1054815.172861   683224.633686
#Sta/Elev= 30
       0 1478.48   14.54 1478.25   26.92 1473.16   39.64 1472.28   63.48 1472.87
  150.32 1469.91  210.18 1466.74  256.96 1465.24  308.63 1464.21  363.15 1463.85
  399.11 1462.48  411.27  1461.5  420.05 1460.05  428.51 1455.95  436.89  1455.1
  453.88 1457.57  479.12 1462.83  506.48 1464.14  522.96 1469.31  540.71 1480.59
   563.6 1498.37   573.9 1505.85  606.93 1526.22  615.69 1532.27   639.8 1546.34
  649.87 1551.52  663.85 1557.75  671.33 1559.63  725.42 1569.66  744.63 1569.38
#Mann= 3 , 0 , 0
       0    .085       0  420.05    .049       0  453.88     .12       0
Bank Sta=420.05,453.88
Exp/Cntr=0.3,0.1

Type RM Length L Ch R = 1 ,4345.773,515.02,501.6,489.58
XS GIS Cut Line= 3
  1054313.045152   684011.358033  1054814.892115    683681.71344
  1055075.655744   683470.150515
#Sta/Elev= 30
       0 1485.75   38.32 1479.25   54.43 1479.57    92.2 1472.94  126.38 1470.66
  210.98 1468.37  265.89 1465.54  428.67 1464.07  466.36 1462.16  583.19 1463.26
  584.83 1461.04  591.62 1452.73  600.18 1452.55  616.79 1454.86  620.34  1456.7
  631.71 1459.24  645.11 1460.72   660.1  1463.9  670.92 1467.53  683.05 1475.99
  692.09 1479.57  715.65 1491.83  766.38 1519.44  774.93 1524.89  801.94 1538.14
  832.69 1556.71  844.74  1566.1  892.16 1595.21  905.66 1600.57  936.22 1608.85
#Mann= 3 , 0 , 0
       0    .085       0  584.83    .049       0  616.79     .12       0
Bank Sta=584.83,616.79
Exp/Cntr=0.3,0.1

Type RM Length L Ch R = 1 ,3844.177,725.03,724.09,704.14
XS GIS Cut Line= 3
  1054611.201316   684497.952796  1055083.527871   684114.187463
  1055334.451352   683691.061573
#Sta/Elev= 30
       0 1489.62    8.56 1489.03   19.52 1486.24   34.37 1479.71   48.79 1477.88
  129.05 1479.28  225.96  1473.2  473.63 1464.33  565.42 1459.52  642.22 1459.95
  679.01 1458.55  685.83 1453.85  695.57 1452.34  703.68 1453.39  710.88 1456.55
  712.74 1458.34   770.9 1458.75  897.52 1462.15  912.27  1470.9  917.69 1475.79
  927.62 1482.18   958.8 1506.34   981.6 1521.78 1009.52 1542.27 1016.89 1546.08
 1024.67 1552.41 1064.08 1579.46 1070.91 1584.47 1084.07 1597.16 1100.51 1604.23
#Mann= 3 , 0 , 0
       0    .085       0  679.01    .049       0  712.74     .09       0
Bank Sta=679.01,712.74
Exp/Cntr=0.3,0.1

Type RM Length L Ch R = 1 ,3120.083,817.75,818.14,791
XS GIS Cut Line= 2
  1055354.131611   685215.298766  1055969.140167   683847.519767
#Sta/Elev= 30
       0 1490.41   21.41 1490.42   67.92 1488.46  176.95 1480.23  227.28  1477.2
  286.52 1474.79  371.41 1469.22   512.6 1461.67  536.11 1461.07  764.75 1460.21
  851.04 1456.93  885.03 1456.63   920.8 1457.16  928.84 1456.25  937.38 1454.44
  941.31 1453.23  954.67 1451.54  962.86 1452.56  971.22 1454.86  995.86 1456.97
 1079.46 1456.08 1268.22    1459 1294.18 1460.46 1317.13 1462.69 1327.76 1465.82
 1340.03  1470.4 1389.21 1493.08 1399.86 1496.24 1434.74 1510.55 1499.68 1532.32
#Mann= 3 , 0 , 0
       0    .085       0  937.38    .049       0  971.22     .09       0
Bank Sta=937.38,971.22
Exp/Cntr=0.3,0.1

Type RM Length L Ch R = 1 ,2301.944,684.83,665.2,635.21
XS GIS Cut Line= 2
  1056234.823871   685396.849269  1056520.187834   684102.871307
#Sta/Elev= 30
       0 1501.51   34.71  1500.2  118.41 1494.03  177.14 1486.64   344.4 1471.92
  462.23  1460.1  553.39 1455.94  706.81 1454.33  717.74 1452.27   724.3  1449.9
  731.56 1448.93  747.84 1451.57  777.52 1452.77  793.37  1454.9  812.53    1455
  838.75 1453.46   880.4 1455.03  888.28 1458.52  939.14 1474.42  990.82 1484.54
  998.25 1487.38 1037.89 1495.32 1059.39  1498.1 1074.68 1498.41 1112.17 1502.49
 1156.67 1504.87 1201.73 1501.36 1248.62 1501.72 1275.55 1507.28 1325.07 1521.37
#Mann= 3 , 0 , 0
       0    .085       0  717.74    .049       0  747.84     .12       0
Bank Sta=717.74,747.84
Exp/Cntr=0.3,0.1

Type RM Length L Ch R = 1 ,1636.742,773.82,778.91,772.68
XS GIS Cut Line= 3
  1057217.438193   686499.619265  1057061.395352   684678.519307
  1056820.311981   684206.192752
#Sta/Elev= 30
       0 1485.86   45.61 1489.04  171.43 1485.61  372.52 1488.78  504.27 1486.88
  627.81 1479.71  644.38 1475.09  666.97 1475.68   703.9 1469.17  785.05 1461.82
  948.43 1466.35 1029.42  1473.5 1043.53 1469.92 1092.57 1477.34 1114.52  1475.4
    1176 1476.69 1237.94 1473.57    1345 1462.71  1492.3 1456.09 1710.42 1451.79
 1928.16  1453.3 1942.91 1449.96 1962.52 1447.17 1981.72 1450.69  1995.1  1454.1
 2115.84 1456.88 2193.48 1464.84 2254.42  1482.6 2323.69 1512.43 2358.07 1521.81
#Mann= 3 , 0 , 0
       0    .085       0 1942.91    .049       0 1981.72    .085       0
Bank Sta=1942.91,1981.72
Exp/Cntr=0.5,0.3

Type RM Length L Ch R = 1 ,857.834 ,135.59,160.06,166.79
BEGIN DESCRIPTION:
Upstream xs of Bridge 37111-0247
END DESCRIPTION:
XS GIS Cut Line= 5
  1058198.509166   685864.421386  1057534.620149   684257.105238
   1057490.83798   684121.004799   1057392.43661   683884.841503
  1057289.945909   683869.502504
#Sta/Elev= 30
   -1340 1534.29-1281.53 1527.95-1238.37 1530.41-1157.99 1559.44-1087.23 1575.32
-1049.96 1577.56  -951.5 1571.28 -924.78  1578.4 -846.81  1588.1 -771.74 1567.79
 -704.41 1563.23 -685.93  1563.7 -609.67 1580.03 -558.89 1584.49 -366.38 1559.18
 -302.34 1541.99 -216.44 1533.34 -124.88 1507.99     108  1472.3   313.2  1457.2
   338.9  1452.2     620  1448.5     637  1441.9     654  1441.3     666  1447.5
   682.2  1453.6   749.9  1456.7   775.2  1465.7     816  1490.5   878.9  1512.2
#Mann= 3 , 0 , 0
   -1340    .085       0     620    .049       0     666     .12       0
#XS Ineff= 2 , 0
       0  558.96 1452.62               0
Permanent Ineff=
       F       F
Bank Sta=620,666
Exp/Cntr=0.5,0.3
